--- Greenbrier Fork.prj (project) ---

Proj Title=Greenbrier Fork
Current Plan=p01
Default Exp/Contr=0,0
English Units
Geom File=g01
Flow File=f01
Plan File=p01
BEGIN DESCRIPTION:
END DESCRIPTION:
DSS Export Rating Curves= 0
DSS Export Rating Curve Sorted= 0
DSS Export Volume Flow Curves= 0
DXF OffsetX= 0
DXF OffsetY= 0
DXF ScaleX= 0
DXF ScaleY= 0

--- Greenbrier Fork.p01 (plan) ---

Plan Title=Floodplain
Program Version=4.00
Geom File=g01
Flow File=f01
K Sum by GR=0
Std Step Tol=0.01
Critical Tol=0.01
Num of Std Step Trials=20
Max Error Tol=0.3
Flow Tol Ratio=0.001
Split Flow NTrial=30
Split Flow Tol=0.02
Split Flow Ratio=0.02
Log Output Level=0
Friction Slope Method=1
Unsteady Friction Slope Method=2
Unsteady Bridges Friction Slope Method=1
Global Log Level=0
CheckData=False
Run HTab=0
Run UNet=0
Run PostProcess=0
UNET Theta=0
UNET Theta Warmup=0
UNET ZTol=0
UNET ZSATol=0
UNET MxIter=0
UNET MaxInSteps=0
UNET DtIC=0
UNET DtMin=0
UNET MaxCRTS=0
UNET WFStab=0
UNET SFStab=0
UNET WFX=0
UNET SFX=0
UNET DSS MLevel=0
UNET DZMax Abort=0
UNET Convert EG Bridges=0
UNET Use Existing IB Tables=0
UNET Froude Limit=0
UNET Froude Power=0
Write IC File=0
Echo Input=False
Echo Output=False
Write Detailed=0

--- Greenbrier Fork.f01 (steady flow) ---

Flow Title=NFF Regression Equation
Program Version=4.00
Number of Profiles=1
Profile Names=P100yr
River Rch & RM=Greenbrier Fork,Main      ,13223.7
525.0549
River Rch & RM=Greenbrier Fork,Main      ,13223.7
577.9099
River Rch & RM=Greenbrier Fork,Main      ,12559.1
628.5913
River Rch & RM=Greenbrier Fork,Main      ,10717.7
656.1679
River Rch & RM=Greenbrier Fork,Main      ,9443
723.3410
River Rch & RM=Greenbrier Fork,Main      ,6870.2
799.5771
River Rch & RM=Greenbrier Fork,Main      ,4475.8
879.9222
River Rch & RM=Greenbrier Fork,Main      ,4175.2
1024.941
River Rch & RM=Greenbrier Fork,Main      ,3302.1
1041.036
River Rch & RM=Greenbrier Fork,Main      ,286.1
1156.141
Boundary for River Rch & Prof#=Greenbrier Fork,Main      ,1
Up Type=0
Dn Type=3
Dn Slope=0.032645

--- Greenbrier Fork.g01 (geometry) ---

Geom Title=USGS 10m DEM
Program Version=4.00

River Reach=Greenbrier Fork ,Main
Reach XY= 30
     1697455.587      168793.166      1697479.42      169028.073
     1697378.184      169288.309     1697404.369      169611.029
     1697672.757      170532.059     1697632.826      170693.091
      1697701.56      170783.427     1698006.605      170954.279
     1698522.434      171030.867     1698767.256      170886.855
     1699070.338      170848.887     1699947.509      170954.933
     1700101.996      170924.821     1700658.641      171044.898
     1701338.837      171715.938     1701587.911      172060.632
     1701908.173      172223.698     1702092.661       172492.42
     1702687.117      173001.955     1703367.094      173091.064
     1703521.988      173409.822     1704444.327      173858.012
     1704669.308       173903.47     1704875.323      173845.591
     1705021.401      173965.863     1705561.563      174212.621
     1706110.554      174269.756     1706318.215      174346.594
     1706834.676      174877.745     1707036.368      174923.976

Type RM Length L Ch R = 1 ,13223.7 ,73.8,73.2,72.6
XS GIS Cut Line= 4
      1696973.66      168802.773     1697365.387      168802.843
     1697535.716      168810.585     1697878.953       168792.52
#Sta/Elev= 30
      10 1526.09    50.2 1508.84   100.4 1488.77   120.5 1481.43   150.7 1472.83
   160.7 1468.95   170.8 1463.22   180.8 1456.27   271.2 1391.82   301.3 1370.94
   331.5 1350.83   361.6 1331.63   381.7 1320.42   421.8 1301.01     472 1280.84
     482 1277.27     487 1276.59     492 1275.91     497 1276.04   502.1 1276.18
   522.1 1278.93   552.2 1281.82   643.1 1291.82     724  1304.2   744.2 1307.69
   754.3 1309.95   774.5 1315.93   784.6 1319.98   804.9 1329.72   905.9 1366.01
#Mann= 3 , 0 , 0
       0     .06       0     487    .045       0     497     .06       0
Bank Sta=487,497
XS Rating Curve= 0 ,0
Exp/Cntr=0.3,0.1

Type RM Length L Ch R = 1 ,13150.5 ,370.8,378,385.2
XS GIS Cut Line= 4
     1696971.491      168878.492     1697402.134      168876.835
      1697605.86      168883.461     1697899.028      168880.148
#Sta/Elev= 30
      10 1548.71      30 1545.92    50.1 1538.72   160.2 1489.19   170.3 1483.35
   180.3 1476.09   220.3 1442.75   240.4  1427.5   270.4  1405.9   290.4 1392.64
   360.5 1350.48   440.4 1306.17   459.8 1294.19   479.2 1279.42   488.9  1274.9
   493.6 1274.54   498.6 1274.14   503.6  1274.9   527.7 1278.96   624.8 1289.38
   674.9 1298.34   705.2 1305.88   735.6  1317.9   796.2 1347.63   826.6  1364.1
   836.7 1370.44   856.9 1385.95     867 1391.34   897.3 1403.62   927.7 1413.42
#Mann= 3 , 0 , 0
       0     .06       0   493.6    .045       0   503.6     .06       0
Bank Sta=493.6,503.6
XS Rating Curve= 0 ,0
Exp/Cntr=0.3,0.1

Type RM Length L Ch R = 1 ,12772.5 ,223.3,213.4,203.5
XS GIS Cut Line= 4
     1696947.541      169148.726     1697325.943      169208.099
     1697536.733      169294.586     1697847.661      169340.728
#Sta/Elev= 30
    10.1 1371.83    40.3 1367.24   151.2 1352.91   181.4 1348.42   191.5 1346.67
   201.6 1344.37   241.9  1334.2   312.5 1317.21   332.6 1311.72   352.8 1304.89
     383 1293.24   422.7  1275.8   442.5 1266.38   447.4 1265.39   452.4 1264.39
   457.4 1264.65   482.1 1266.82     492 1268.28   511.8 1273.36   561.3 1288.49
   581.2 1293.51     601 1297.85   650.2 1307.37   669.8 1312.08   718.9 1328.17
   758.2 1342.12   817.2 1362.33   846.6 1373.46   885.9 1387.47   925.2 1402.68
#Mann= 3 , 0 , 0
       0     .06       0   447.4    .045       0   457.4     .06       0
Bank Sta=447.4,457.4
XS Rating Curve= 0 ,0
Exp/Cntr=0.3,0.1

Type RM Length L Ch R = 1 ,12559.1 ,342.1,340,337.9
XS GIS Cut Line= 4
     1697061.735      169417.955     1697310.829       169453.54
     1697553.454       169427.66     1697851.073      169411.485
#Sta/Elev= 30
    10.1 1312.54    40.3 1311.12    50.3 1310.07   130.8 1299.46     161 1293.65
   181.2 1288.67   191.2 1285.74   211.4 1278.46   221.4 1275.53   231.5 1273.48
   261.4 1268.65   300.4  1263.6   329.7 1258.34   334.5 1258.14   339.5 1257.93
   344.5 1258.38     359 1260.47   368.7 1262.81   417.5 1276.47   456.6 1286.16
   485.9 1294.57   525.4 1307.53   535.4 1311.48   555.2 1320.87   604.9 1349.73
   634.7 1365.23   684.4  1389.7   714.2 1403.01   753.9 1418.25   793.7 1435.35
#Mann= 3 , 0 , 0
       0     .06       0   334.5    .045       0   344.5     .06       0
Bank Sta=334.5,344.5
XS Rating Curve= 0 ,0
Exp/Cntr=0.3,0.1

Type RM Length L Ch R = 1 ,12219.1 ,249.1,247.9,246.6
XS GIS Cut Line= 4
     1697029.341      169882.027     1697362.589      169784.173
     1697614.737      169733.507     1697927.043       169706.99
#Sta/Elev= 30
     9.9 1497.21    59.5 1469.39   148.9 1421.16   158.8 1415.21   168.7 1408.54
   198.5 1387.26   287.8 1322.16   297.7  1315.5   307.6 1309.99   347.3  1293.6
   406.7 1264.34   416.6 1260.15   426.5 1257.48   456.1 1252.16     461 1251.65
     466 1251.12     471 1251.41   475.9 1251.69   485.8 1254.17   564.9 1285.83
   614.6 1304.83   665.2 1326.55   685.4 1336.92   705.6    1348   725.8 1359.72
   746.1 1372.24   766.3 1385.58   806.7 1413.95   877.5 1465.43   917.9 1493.34
#Mann= 3 , 0 , 0
       0     .06       0     461    .045       0     471     .06       0
Bank Sta=461,471
XS Rating Curve= 0 ,0
Exp/Cntr=0.3,0.1

Type RM Length L Ch R = 1 ,11971.2 ,229,230.6,232.3
XS GIS Cut Line= 4
     1697107.024      170072.088     1697420.819      170030.033
     1697699.028      169955.628     1697980.473      169952.393
#Sta/Elev= 30
     9.9  1448.7    39.6 1428.79   108.8  1387.5   158.3 1356.34   197.9 1330.73
   217.7 1318.95   237.4 1309.53   267.1 1298.05   286.9 1292.13   306.7 1287.49
   326.5  1282.1   356.3 1271.95   376.2 1263.65     396 1253.74     406 1249.67
   410.9  1248.9   415.9 1248.11   420.9 1248.56   425.8    1249   445.7 1254.68
   564.9  1298.2   604.6 1314.02   634.7 1327.81   664.9 1343.68     685 1355.39
   715.2 1374.36   765.4 1406.92   805.6  1431.7   845.8 1454.84     886 1476.67
#Mann= 3 , 0 , 0
       0     .06       0   410.9    .045       0   420.9     .06       0
Bank Sta=410.9,420.9
XS Rating Curve= 0 ,0
Exp/Cntr=0.3,0.1

Type RM Length L Ch R = 1 ,11740.6 ,476.1,475.2,474
XS GIS Cut Line= 4
     1697149.424       170318.09     1697466.109      170243.542
     1697708.495       170200.37     1698041.107      170129.485
#Sta/Elev= 30
     9.9  1483.9    49.3 1452.33    88.7 1422.11   256.3 1306.79     276 1294.06
   285.9 1288.85   295.8 1285.19   305.6  1283.5   354.9  1282.6   364.7 1281.14
   374.6 1277.93   384.4 1273.34     414 1257.79   423.8 1251.51   433.7 1246.93
   438.5 1246.53   443.5 1246.12   448.5 1247.54   453.4 1248.92   502.6 1274.45
   512.5 1278.24   522.3 1280.53   561.7 1285.01   571.5  1287.9   581.5 1292.39
   651.6 1335.93   721.6 1375.97   811.6 1432.92   871.6 1464.78   911.6 1484.65
#Mann= 3 , 0 , 0
       0     .06       0   438.5    .045       0   448.5     .06       0
Bank Sta=438.5,448.5
XS Rating Curve= 0 ,0
Exp/Cntr=0.3,0.1

Type RM Length L Ch R = 1 ,11265.4 ,569.7,547.7,525.9
XS GIS Cut Line= 4
     1697275.796      170950.651     1697540.513      170696.441
     1697747.715      170641.745     1698112.097      170444.186
#Sta/Elev= 30
     9.9 1416.61    39.7 1399.26   109.1 1364.17     129 1351.98   178.5 1316.87
   188.5 1311.08   198.4 1306.99   208.3 1305.06     248 1301.58   267.8 1297.77
   287.7 1291.65   307.5 1284.15   317.4 1279.84   337.3 1269.08   347.2 1266.18
     367 1263.16   425.5 1249.21   454.7 1238.47   459.4 1237.64   464.4 1236.76
   469.4 1236.81   513.1  1240.8   552.1 1242.47   571.6 1245.45   591.4 1252.76
   682.4 1291.24   702.6  1302.6   834.1 1386.63   935.1  1453.3   995.8 1489.49
#Mann= 3 , 0 , 0
       0     .06       0   459.4    .045       0   469.4     .06       0
Bank Sta=459.4,469.4
XS Rating Curve= 0 ,0
Exp/Cntr=0.3,0.1

Type RM Length L Ch R = 1 ,10717.7 ,257,252.5,248
XS GIS Cut Line= 4
     1697893.128        171395.2     1698025.763      171074.935
     1698083.982      170848.481     1698219.783      170526.283
#Sta/Elev= 30
     9.9 1374.82    19.8  1364.4    29.7 1360.04    39.6 1358.06    49.5 1355.14
    59.4 1351.25    89.1 1338.32   138.7  1315.1   168.4 1301.88   198.1 1289.83
   227.8  1279.5   277.3 1264.19   326.8 1251.43   366.1 1243.04   444.1 1228.42
   458.6 1227.07   463.6 1226.95   468.6 1227.47   473.3 1227.97     483 1230.95
   531.7 1255.58   610.4 1294.03   760.3 1362.57   770.3 1368.35   780.3 1375.22
   820.2 1405.67   850.2 1429.73   870.2 1444.93   880.2 1451.69   930.1 1483.16
#Mann= 3 , 0 , 0
       0     .06       0   458.6    .045       0   468.6     .06       0
Bank Sta=458.6,468.6
XS Rating Curve= 0 ,0
Exp/Cntr=0.3,0.1

Type RM Length L Ch R = 1 ,10465.2 ,280.9,273.8,266.6
XS GIS Cut Line= 4
     1698126.047      171443.725     1698297.502       171104.05
     1698303.972      170916.421     1698355.732      170625.271
#Sta/Elev= 30
      10 1379.33    60.1  1366.5    70.1 1363.03    80.1 1358.37    90.1 1352.68
   110.1 1339.51   120.2 1333.94   190.2 1303.68   240.3 1285.31   260.3 1279.39
   290.4 1271.69   330.4 1264.58   360.5 1257.32   380.5 1251.63   410.1    1241
   439.8  1232.7   479.3 1225.58   484.2 1225.24   489.2 1224.89   494.2 1225.35
   499.1  1225.8   508.9 1228.67   528.7 1238.38   568.2 1261.92   637.2 1301.43
   725.9 1342.01   785.1 1367.35   794.9 1372.74   824.5 1392.16   863.9 1416.44
#Mann= 3 , 0 , 0
       0     .06       0   484.2    .045       0   494.2     .06       0
Bank Sta=484.2,494.2
XS Rating Curve= 0 ,0
Exp/Cntr=0.3,0.1

Type RM Length L Ch R = 1 ,10191.5 ,485.4,489.5,493.7
XS GIS Cut Line= 4
     1698590.326      171475.484     1698604.826       171129.93
     1698543.361      170942.301      1698408.02      170561.023
#Sta/Elev= 30
     9.9 1453.58    29.6 1441.05    59.3 1419.09    88.9 1398.87   138.3 1367.08
   158.1 1357.19   187.8 1346.81   197.6    1342   207.5 1334.72   227.3 1315.25
   237.2 1308.95   286.6 1287.52   345.9 1258.89   434.7 1224.03   439.6 1222.74
  444.59 1221.35   449.6 1221.42   454.5 1221.43   464.3 1223.87   533.4 1248.63
   583.8 1263.85   614.1 1275.08   634.3 1284.07     695 1314.57   745.6 1342.44
   796.2 1365.42   816.4 1375.47   836.6 1387.54   877.1 1414.53   947.9 1459.47
#Mann= 3 , 0 , 0
     9.9      .1       0   439.6    .045       0   449.6      .1       0
Bank Sta=439.6,449.6
XS Rating Curve= 0 ,0
Exp/Cntr=0.3,0.1

Type RM Length L Ch R = 1 ,9701.9  ,252.4,258.9,265.4
XS GIS Cut Line= 4
     1699001.776      171315.393     1699018.905      170961.711
     1698993.025      170715.851     1698942.918      170406.846
#Sta/Elev= 30
     9.8 1389.04    68.9 1346.44   127.9 1301.16   147.5  1288.3   157.4 1283.66
   167.2 1281.02   196.7 1277.71   216.4 1273.44   285.2 1249.22     364  1224.1
   383.8 1219.71   423.3  1213.3     453 1206.08   457.9 1205.58   462.9 1205.08
   467.9 1205.32   472.8 1205.56   482.6 1208.09   502.4 1215.38   532.1 1224.11
   551.9 1228.19   591.4 1234.13   601.3 1237.04   621.5 1244.75   631.6 1247.57
   722.5 1264.69   752.8  1269.1   762.9 1271.37   813.4 1287.36   914.4 1326.45
#Mann= 3 , 0 , 0
       0      .1       0   457.9    .045       0   467.9      .1       0
Bank Sta=457.9,467.9
XS Rating Curve= 0 ,0
Exp/Cntr=0.3,0.1

Type RM Length L Ch R = 1 ,9443    ,239.9,227.1,214.3
XS GIS Cut Line= 4
     1699154.775      171294.915     1699245.355      170955.241
     1699284.175      170780.551     1699251.825      170469.992
#Sta/Elev= 30
      10 1380.56    50.2 1358.23   100.4 1329.06   140.6 1306.38     221 1264.55
     231 1260.18   241.1  1256.7   291.3 1241.34   341.5 1225.25   401.3 1206.83
   411.2 1203.49   421.1 1200.48   426.1  1199.8   431.1 1199.13   436.1 1199.98
     441  1200.8     451 1205.58   470.8 1217.76   510.6 1239.82   570.8 1271.96
     601 1287.18   611.1 1291.14   681.6 1312.13   711.8 1322.33   762.2 1342.46
   782.3 1351.15   812.5 1364.87   822.6 1368.37   832.7 1370.35   842.7 1371.28
#Mann= 3 , 0 , 0
       0      .1       0   426.1    .045       0   436.1      .1       0
Bank Sta=426.1,436.1
XS Rating Curve= 0 ,0
Exp/Cntr=0.3,0.1

Type RM Length L Ch R = 1 ,9215.9  ,119,133.3,147.6
XS GIS Cut Line= 4
     1699527.532      171356.103     1699513.859      170974.651
     1699439.454      170806.431     1699413.648      170432.084
#Sta/Elev= 30
      10 1332.12    50.2 1319.64   100.4 1305.44   180.8 1286.02     221 1275.19
   241.1  1268.6   281.3 1250.46   291.3 1247.13   311.4 1244.37   331.5 1240.41
   351.6 1235.09   371.7 1228.61   420.4 1208.08   449.5 1196.98   454.1    1196
   459.1 1194.94   464.1 1195.04   468.8 1195.13   478.5  1197.4   507.6 1208.54
   536.6 1220.98   565.6 1235.32   634.8 1275.29   674.3 1296.13   703.9 1309.18
   753.3 1328.87   802.6 1351.28   832.3 1367.51   901.4 1409.18   940.9 1433.97
#Mann= 3 , 0 , 0
       0      .1       0   454.1    .045       0   464.1      .1       0
Bank Sta=454.1,464.1
XS Rating Curve= 0 ,0
Exp/Cntr=0.3,0.1

Type RM Length L Ch R = 1 ,9082.6  ,127.3,125.3,123.2
XS GIS Cut Line= 4
     1699559.149       171220.51     1699581.794      170958.476
     1699630.319      170780.551     1699594.734      170469.992
#Sta/Elev= 30
     9.7 1292.63    48.7 1282.21    87.7 1270.31   116.9 1259.67   146.1 1246.92
   155.9 1244.03   204.6 1242.66   214.3 1241.63     224 1239.64   233.8 1236.51
   243.5 1232.41   292.1 1208.63   311.5 1197.54   316.2 1195.93   321.2 1194.23
   326.2 1194.33     331 1194.43   340.7 1197.83   360.1 1208.05   398.9    1226
   418.3 1235.93   477.7 1270.77   528.1 1298.91   568.4 1319.96   588.6 1332.42
   628.9 1359.63   649.1 1371.11   719.7 1408.93   739.9 1420.58     760 1433.18
#Mann= 3 , 0 , 0
       0      .1       0   316.2    .045       0   326.2      .1       0
Bank Sta=316.2,326.2
XS Rating Curve= 0 ,0
Exp/Cntr=0.3,0.1

Type RM Length L Ch R = 1 ,8957.3  ,226.2,223.8,221.5
XS GIS Cut Line= 4
     1699575.324        171330.5     1699707.959      171000.531
     1699743.544      170787.021     1699746.779      170476.462
#Sta/Elev= 30
     9.9 1325.79    39.5 1321.13   138.3 1291.27   197.6 1269.43   266.7 1241.33
   276.6 1237.85   286.5 1235.81   306.2 1234.62   316.1 1232.68     326 1229.53
   355.6 1216.24     395 1201.91   414.7 1193.39   419.5 1191.99   424.5 1190.52
   429.5 1190.53   434.3 1190.54   444.2 1192.74   463.9 1199.05   493.4 1209.75
   532.7 1225.97   552.4  1236.6   592.1 1262.88   632.2 1286.56   652.2 1299.56
   672.3 1314.45   732.4 1363.27   762.4  1385.4   822.5 1424.09   882.7 1461.68
#Mann= 3 , 0 , 0
       0     .06       0   419.5    .045       0   429.5     .06       0
Bank Sta=419.5,429.5
XS Rating Curve= 0 ,0
Exp/Cntr=0.3,0.1

Type RM Length L Ch R = 1 ,8733.5  ,501.7,498.9,496.1
XS GIS Cut Line= 4
     1699841.998      171395.077     1699934.408      171081.405
     1699944.113      170864.661     1699945.106      170482.936
#Sta/Elev= 30
     9.9 1389.32    69.4 1354.72   118.9 1327.58   158.5 1305.27   178.4 1293.35
     218 1268.07   227.9 1262.32   247.7 1251.79   317.1 1221.23     327 1217.28
   336.9 1214.32   356.6 1209.39   386.2 1200.12   425.6 1188.49   445.3 1182.06
   450.2 1181.72   455.2 1181.38   460.2 1182.47   465.1 1183.55   474.9 1187.95
   484.8 1192.85     544 1220.15   594.2 1245.25   664.5 1281.11   674.6  1286.8
   704.7 1304.94   754.9 1333.47   825.2 1374.71   845.3 1387.59   925.7 1441.94
#Mann= 3 , 0 , 0
       0     .06       0   450.2    .045       0   460.2     .06       0
Bank Sta=450.2,460.2
XS Rating Curve= 0 ,0
Exp/Cntr=0.3,0.1

Type RM Length L Ch R = 1 ,8234.6  ,491.3,511.7,532.2
XS GIS Cut Line= 4
     1700357.409      171462.188     1700429.362      171120.225
     1700406.717      170884.071     1700451.371      170543.149
#Sta/Elev= 30
      10 1400.77    39.9 1380.99    89.9  1343.7   119.8 1323.57   139.8 1311.22
   289.5 1224.14   329.5 1197.51   349.5  1186.1   359.3 1182.15   369.2 1179.09
   379.1 1176.95     389 1175.74   398.9 1175.45   438.4 1175.92   458.2  1172.2
   463.1 1172.12   468.1 1172.03   473.1 1173.09   497.7 1180.38   517.5 1187.78
   566.9 1210.67     617 1232.42   627.1 1237.38   687.8 1270.49   728.3 1291.38
   788.9 1328.39   859.7 1368.87   890.1 1387.05   910.3 1397.82   930.5 1407.73
#Mann= 3 , 0 , 0
       0     .06       0   463.1    .045       0   473.1     .06       0
Bank Sta=463.1,473.1
XS Rating Curve= 0 ,0
Exp/Cntr=0.3,0.1

Type RM Length L Ch R = 1 ,7722.9  ,498.9,496.7,494.5
XS GIS Cut Line= 4
     1700478.397      171526.784     1700749.627       171298.15
     1700950.196      171146.105     1701183.887      170943.917
#Sta/Elev= 30
     9.9  1393.6    59.1  1362.4   128.1 1317.59     138 1311.77   157.7 1301.14
   197.1 1277.94   256.2 1241.83     335 1192.16   364.8 1174.26   374.9 1168.62
   384.9 1164.31     395 1162.11   425.2 1160.06   445.3 1157.39   450.4 1157.19
   455.4 1156.99   460.4 1157.98   465.5 1158.99   475.5 1162.78     536 1187.36
   556.1 1193.32   566.2 1196.75   576.2 1201.04   616.4 1222.38   716.1 1273.54
   765.9  1301.1   835.7 1342.06   845.7 1348.36   865.6 1361.94   915.4 1398.66
#Mann= 3 , 0 , 0
       0     .06       0   450.4    .045       0   460.4     .06       0
Bank Sta=450.4,460.4
XS Rating Curve= 0 ,0
Exp/Cntr=0.3,0.1

Type RM Length L Ch R = 1 ,7226.2  ,350.3,356,361.7
XS GIS Cut Line= 4
     1700917.063      171925.015     1701102.241      171660.469
     1701293.105       171479.31     1701513.165      171233.214
#Sta/Elev= 30
    10.1 1244.88    60.5 1233.16   131.2 1218.86     222 1203.49   252.3 1195.04
   282.6 1184.77   292.6 1180.51   322.9 1165.88   352.2 1155.81   371.6 1151.44
   381.4 1149.94   410.6 1147.51   434.9 1144.28   439.9 1143.65   444.9  1143.7
   449.6 1143.75   459.4 1147.77   478.9  1163.8   488.6 1170.75   498.4 1176.66
   508.1  1180.8   547.1 1192.46   606.1 1216.19   666.1 1237.49   676.1 1240.76
   696.1 1245.85   716.1 1252.64   826.2 1293.92   886.2 1314.52   916.2 1327.08
#Mann= 3 , 0 , 0
       0     .06       0   434.9    .045       0   444.9     .06       0
Bank Sta=434.9,444.9
XS Rating Curve= 0 ,0
Exp/Cntr=0.3,0.1

Type RM Length L Ch R = 1 ,6870.2  ,265,255.9,246.8
XS GIS Cut Line= 4
     1701001.956      172009.848     1701338.395      171886.919
     1701551.905      171776.929     1701710.419      171495.485
#Sta/Elev= 30
     9.9 1256.98    39.8 1257.58    49.7  1256.4    59.7 1253.21    89.5 1238.56
    99.5 1234.41   179.1 1205.11   208.9 1193.25   248.7 1175.24   278.6 1158.96
   288.5 1154.34   318.4 1142.84   328.3  1140.2   338.3 1138.67   408.2  1135.3
   443.3 1132.11   448.3 1131.94   453.3 1133.17   458.3 1134.41   468.3 1141.28
   478.3 1149.25   498.3 1162.86   598.4 1225.38   638.7 1253.53   679.1 1280.29
   739.7 1317.27   759.9 1327.15   830.5 1356.93   860.8 1370.45   921.4 1399.96
#Mann= 3 , 0 , 0
       0     .06       0   443.3    .045       0   453.3     .06       0
Bank Sta=443.3,453.3
XS Rating Curve= 0 ,0
Exp/Cntr=0.3,0.1

Type RM Length L Ch R = 1 ,6614.3  ,407.4,410.3,413.1
XS GIS Cut Line= 4
     1701089.807      172162.612     1701513.085      172129.543
      1701665.13      171925.739     1701849.103      171654.163
#Sta/Elev= 30
    10.1  1331.8    30.3 1324.43    60.7 1312.28   161.7 1267.97   202.2 1250.82
   222.4 1241.43     283 1211.06   333.6 1189.04     374 1172.81   424.6  1153.5
   473.5 1131.28   483.2 1127.68   502.8 1123.66   517.4 1122.31   522.4 1122.23
   527.4 1123.16   532.1 1124.03     581  1142.7   590.8 1146.93   669.1 1185.96
   728.5 1214.15   778.2  1240.4   808.1 1257.47   847.8 1281.38   857.8 1288.91
   877.6 1307.41   887.6 1315.68   957.2 1357.71     987 1377.05  1006.9 1390.87
#Mann= 3 , 0 , 0
       0     .06       0   517.4    .045       0   527.4     .06       0
Bank Sta=517.4,527.4
XS Rating Curve= 0 ,0
Exp/Cntr=0.3,0.1

Type RM Length L Ch R = 1 ,6204    ,439.3,438.7,438.1
XS GIS Cut Line= 4
     1701583.306      172566.405     1701852.759      172320.408
     1702046.859      172126.308     1702159.002      171837.557
#Sta/Elev= 30
     9.9  1306.7   118.3 1236.81   147.9 1218.29   177.5 1200.52   197.2 1189.18
   216.9 1178.44   246.5 1163.68   276.1 1150.09   335.3 1125.06   345.1 1122.01
     355 1120.28   433.5 1114.75   457.9 1111.61   462.9 1111.14   467.9 1111.56
   472.7 1111.96   482.5 1115.51   492.3 1121.69   511.9 1135.38   570.7    1179
   580.5 1185.69   590.3 1191.39   600.1 1196.21   679.3    1229   709.3 1244.09
   759.3 1267.69   819.2 1297.96   849.2 1312.46   909.1 1337.39   949.1 1354.89
#Mann= 3 , 0 , 0
       0     .06       0   457.9    .045       0   467.9     .06       0
Bank Sta=457.9,467.9
XS Rating Curve= 0 ,0
Exp/Cntr=0.3,0.1

Type RM Length L Ch R = 1 ,5765.2  ,509,507.1,505.2
XS GIS Cut Line= 4
     1701920.205      172952.531     1702114.794      172673.022
     1702275.224      172503.186     1702493.153      172245.292
#Sta/Elev= 30
      10 1252.63    40.1 1244.24    70.1 1235.12   110.2 1220.43   130.2 1214.06
   170.3 1197.81   180.3 1193.44   200.3 1183.66   220.4 1174.84   270.5 1157.04
   310.5 1143.87     399 1109.87   408.7 1106.84   437.9 1099.04   442.7 1098.48
   447.7 1097.89   452.7 1098.48   457.4 1099.02   467.1 1104.06   476.9 1111.81
   486.6 1118.92   496.3 1125.36     545 1157.02   623.9 1207.22   663.6 1231.39
   762.9 1292.85   812.5 1322.85   882.1 1364.15     892 1370.38   911.8 1383.57
#Mann= 3 , 0 , 0
       0     .08       0   442.7    .045       0   452.7     .08       0
Bank Sta=442.7,452.7
XS Rating Curve= 0 ,0
Exp/Cntr=0.3,0.1

Type RM Length L Ch R = 1 ,5258.1  ,139.4,136.2,132.9
XS GIS Cut Line= 4
     1702257.283      173212.279     1702506.228      173009.461
     1702695.602       172768.24     1702878.127      172541.281
#Sta/Elev= 30
      10 1263.46    70.2 1230.32    90.3 1220.02   130.4 1201.38   230.8  1158.8
   260.9 1144.38   311.1 1118.02   340.9 1105.75   360.7 1098.82   429.9 1079.95
   434.8 1079.18   439.8 1078.38   444.8  1078.5   459.6 1079.82   479.4  1084.7
   509.1 1095.98   528.9  1104.8   558.5 1120.35   637.8 1167.97     678 1191.42
   708.1 1207.53   738.3 1221.45   758.3 1232.45   788.5 1251.44   808.6 1266.24
   828.6 1282.75   868.8  1318.5   888.9 1334.49   898.9  1341.4     919 1352.68
#Mann= 3 , 0 , 0
       0     .06       0   434.8    .045       0   444.8     .06       0
Bank Sta=434.8,444.8
XS Rating Curve= 0 ,0
Exp/Cntr=0.3,0.1

Type RM Length L Ch R = 1 ,5122    ,124.4,116.4,108.5
XS GIS Cut Line= 4
     1702405.084      173245.937     1702629.408      173100.429
     1702730.455      172918.545     1702841.606      172645.719
#Sta/Elev= 30
     9.9 1253.97    69.3 1228.14      99  1214.4   118.8 1203.43   148.5  1185.6
   178.3 1168.56   237.7 1135.32   267.4 1119.86   287.2 1107.91   297.1 1102.65
     307 1098.75   326.8 1095.29   336.7 1092.56   346.6 1088.63   366.5  1079.4
   376.4 1076.19   381.3 1075.86   386.3 1075.52   391.3 1075.92   435.8 1081.12
   485.3 1086.07   495.1 1089.21   504.9 1093.96   563.8 1126.88   593.3 1144.15
   671.9 1194.32   711.1 1217.91     721 1224.19   740.6 1237.96     770 1261.48
#Mann= 3 , 0 , 0
       0     .06       0   381.3    .045       0   391.3     .06       0
Bank Sta=381.3,391.3
XS Rating Curve= 0 ,0
Exp/Cntr=0.3,0.1

Type RM Length L Ch R = 1 ,5005.5  ,183.5,182.6,181.8
XS GIS Cut Line= 4
     1702506.228      173355.606     1702777.967      173187.386
     1702810.317      172893.001     1702942.952      172579.207
#Sta/Elev= 30
      10 1295.36    39.9 1280.38   119.8 1246.92   179.8 1219.95   229.7 1195.08
   279.6  1167.5   299.6 1159.31   309.6    1151   339.3 1122.95   359.1 1108.23
     369 1102.29   388.7  1095.7   438.1 1085.06   457.8 1074.94   462.7 1074.29
   467.7 1073.61   472.7  1074.8   497.3 1079.25   546.6 1079.77   586.1 1082.67
     596 1083.98   605.9 1087.25   655.8 1117.07     746 1174.73   806.1 1208.09
   826.2  1222.2   856.2 1246.37   886.3 1268.57   926.4  1296.9   956.4 1316.48
#Mann= 3 , 0 , 0
       0     .06       0   462.7    .045       0   472.7     .06       0
Bank Sta=462.7,472.7
XS Rating Curve= 0 ,0
Exp/Cntr=0.3,0.1

Type RM Length L Ch R = 1 ,4822.9  ,255.7,257.1,258.5
XS GIS Cut Line= 4
     1702957.837      173502.471     1702965.597      173187.386
     1702988.242      172838.007     1703042.525      172591.663
#Sta/Elev= 30
     9.8 1183.83    29.5 1173.94    39.4 1172.04    68.9  1177.5    88.6 1179.29
   108.3 1178.45   118.2 1175.93   187.1 1150.66   246.2 1123.93   295.5  1111.6
   345.2 1095.68   385.2 1086.83   440.2 1068.36   445.2 1067.29   450.2  1067.9
   475.2 1075.13   485.2 1075.76   565.3 1070.42   575.3 1070.98   585.3 1073.69
   625.3 1093.67   665.3  1118.6   725.8 1151.55   756.1  1170.8   806.6 1206.54
   826.7 1223.25   846.9 1242.32     857  1249.4   877.2 1256.96   917.5 1266.09
#Mann= 3 , 0 , 0
     9.8     .06       0   440.2    .045       0   450.2     .06       0
#XS Ineff= 2 , 0
                          488.83         1091.28
Permanent Ineff=
       F       F
Bank Sta=440.2,450.2
XS Rating Curve= 0 ,0
Exp/Cntr=0.3,0.1

Type RM Length L Ch R = 1 ,4565.7  ,89.3,89.9,90.1
XS GIS Cut Line= 4
     1703003.281      173429.842     1703207.395      173187.329
     1703247.814      172880.147     1703235.688      172641.677
#Sta/Elev= 30
     9.9 1161.81    69.3 1148.87   118.9 1135.72   178.3 1121.01   217.9 1108.45
   257.5 1092.43   277.4 1085.41     317 1078.08   416.9 1066.17   441.9 1060.18
   446.9 1059.39   451.9 1059.97   456.9 1060.55   476.9 1067.27   486.9 1068.26
   506.9 1067.68   546.9 1064.42   576.8 1063.73   586.8 1064.33   616.8 1067.98
   656.7 1070.25   666.6 1071.67   676.6 1075.01   716.3 1096.44     776 1123.95
   795.9 1130.75   825.8 1136.84   835.7 1139.67   845.7 1143.44   865.6 1152.34
#Mann= 3 , 0 , 0
       0     .06       0   441.9    .045       0   451.9     .06       0
Bank Sta=441.9,451.9
XS Rating Curve= 0 ,0
Exp/Cntr=0.3,0.1

Type RM Length L Ch R = 1 ,4475.8  ,150.9,170,189.6
XS GIS Cut Line= 4
     1703010.887       173494.71     1703292.331      173171.211
     1703334.386      172928.586     1703467.021      172705.372
#Sta/Elev= 30
      10 1189.04    49.9 1177.49    89.7    1162   159.6 1139.29   189.5 1128.07
   329.1 1083.29   428.8 1062.08   468.2  1056.5   512.4 1054.71   517.4 1054.53
   522.4 1054.68   527.3 1054.82   537.1 1057.63     547 1063.04   556.8 1067.22
   566.7 1067.42   586.4 1063.45   606.1 1064.38   625.8 1069.81   635.6 1070.71
     675 1071.21   744.9 1079.44   764.9 1077.62   784.9 1074.36   794.9 1074.94
   804.9 1076.31   834.8 1083.61   874.8 1091.18   894.7 1093.51   934.7  1096.1
#Mann= 3 , 0 , 0
       0     .06       0   512.4    .045       0   522.4     .06       0
Bank Sta=512.4,522.4
XS Rating Curve= 0 ,0
Exp/Cntr=0.3,0.1

Type RM Length L Ch R = 1 ,4305.8  ,129.7,130.6,131.5
XS GIS Cut Line= 4
     1703052.942       173501.18     1703337.621      173222.971
     1703525.251      173125.921       1703622.3      172795.952
#Sta/Elev= 30
      10 1200.17    19.9 1195.86    69.7 1168.77   139.3 1133.16   159.2 1123.91
   179.1  1117.2   238.8 1099.51   278.6 1088.64   418.2 1054.73   428.2  1052.9
   438.3 1052.11   478.5  1051.1   493.6 1049.96   498.6  1049.5   503.6  1049.7
   508.7 1049.91   518.8  1053.2     559 1077.13   609.3 1105.21   678.1  1132.1
   717.4 1145.76   776.4  1163.2   805.8  1172.6   815.7  1175.2   825.5 1177.01
   835.3 1178.39   874.6 1181.92   913.9  1186.7   933.6 1188.16   953.2 1188.46
#Mann= 3 , 0 , 0
       0     .06       0   493.6    .045       0   503.6     .06       0
Bank Sta=493.6,503.6
XS Rating Curve= 0 ,0
Exp/Cntr=0.3,0.1

Type RM Length L Ch R = 1 ,4175.2  ,245.6,233.6,221.4
XS GIS Cut Line= 4
     1703073.692      173556.866     1703340.856       173352.37
      1703635.24      173216.501      1703842.28      172938.291
#Sta/Elev= 30
     9.9 1229.35    39.6 1217.54    59.4 1206.93    89.1 1189.25   118.7 1170.07
   168.2 1133.26   197.9 1111.97   207.8 1105.76   217.7 1101.36   267.2 1084.52
     287 1078.89   306.8 1075.26   336.4 1073.68   346.3 1072.73   356.1 1070.94
     415 1052.53   444.5 1046.27   459.2 1044.84   464.2 1044.68   469.2 1044.96
   503.5 1049.11   513.3 1050.98   523.1    1055   532.9 1060.23   572.2 1082.55
   621.4 1109.14   660.7 1131.77   868.7 1262.74   898.5 1278.72  1007.5 1333.75
#Mann= 3 , 0 , 0
       0     .06       0   459.2    .045       0   469.2     .06       0
Bank Sta=459.2,469.2
XS Rating Curve= 0 ,0
Exp/Cntr=0.3,0.1

Type RM Length L Ch R = 1 ,3941.5  ,217.2,213.9,210.8
XS GIS Cut Line= 4
     1703279.391       173695.28     1703567.306      173530.295
     1703683.765      173332.961     1703890.805      173054.751
#Sta/Elev= 30
    10.1 1229.77    50.3 1205.64   110.6 1165.18   130.7 1152.91   160.9 1136.94
   221.2 1107.16   261.4 1089.53   331.8 1062.53   341.8 1059.69   381.6 1051.81
   391.6 1049.05   411.5 1041.45   416.5  1041.2   421.5 1040.96   426.5 1042.52
   451.4    1050   481.3 1061.93   531.1 1083.44   580.8 1106.02   600.6 1113.62
   620.4 1123.73   640.2 1135.64     670    1156   699.7  1179.3   739.3 1212.69
   759.1 1228.71   788.9 1251.38   808.7 1265.58   818.6 1271.67   907.8 1321.51
#Mann= 3 , 0 , 0
       0     .06       0   416.5    .045       0   426.5     .06       0
Bank Sta=416.5,426.5
XS Rating Curve= 0 ,0
Exp/Cntr=0.3,0.1

Type RM Length L Ch R = 1 ,3727.6  ,248.9,249.1,249.3
XS GIS Cut Line= 4
     1703669.152      173995.174       1703751.7       173649.99
     1703864.925       173391.19     1703957.234       173131.88
#Sta/Elev= 30
     9.9 1187.14    29.6  1175.5      69 1157.98    88.7 1151.72   197.2 1120.71
   216.9 1113.69   256.3 1097.42   266.2 1094.05   285.9 1089.35   305.6  1087.1
   315.5 1085.05   325.3 1081.91   345.1 1073.98   385.2 1054.84   405.4 1046.08
   435.6 1037.54   450.8 1034.91   455.8 1034.49   460.8 1034.89   526.4 1046.49
   536.5 1049.17   546.6 1053.96   556.7 1060.21     587 1080.45   617.2 1099.37
   627.3 1106.74   765.2 1218.55     834 1271.61   843.8    1278   912.7 1315.68
#Mann= 3 , 0 , 0
       0     .06       0   450.8    .045       0   460.8     .06       0
Bank Sta=450.8,460.8
XS Rating Curve= 0 ,0
Exp/Cntr=0.3,0.1

Type RM Length L Ch R = 1 ,3478.6  ,178.7,176.5,174.2
XS GIS Cut Line= 4
      1703842.28      174012.309      1703978.15       173747.04
     1704062.259       173559.41     1704152.839      173242.381
#Sta/Elev= 30
     9.9 1187.76    59.6 1159.05    69.5 1153.77   139.1 1120.69   208.6 1085.14
   258.3 1062.24   268.2 1058.85   288.1 1054.87     298 1052.02   337.2 1035.84
     347 1032.85     391 1026.74     396  1026.3     401 1026.33   415.5 1027.08
   425.3 1028.43   435.1 1030.41   444.9 1033.44   474.3 1044.66   484.1 1049.04
   553.6 1082.31   563.6 1087.64   573.6 1094.28   583.6 1102.21   653.5  1160.4
   703.5 1203.08   783.4 1269.63   793.4 1277.42   803.4 1284.34   833.4 1300.81
#Mann= 3 , 0 , 0
       0     .06       0     391    .045       0     401     .06       0
Bank Sta=391,401
XS Rating Curve= 0 ,0
Exp/Cntr=0.3,0.1

Type RM Length L Ch R = 1 ,3302.1  ,331,330.7,330.3
XS GIS Cut Line= 4
     1704035.127      174180.453     1704133.429      173847.324
     1704211.069      173607.935     1704367.439      173331.317
#Sta/Elev= 30
     9.9 1202.77    39.7 1188.44    89.3  1167.7     129  1152.8   158.8 1142.97
   188.6 1130.87   267.9 1092.63   347.3 1057.17   387.6 1039.74   407.7 1031.63
   427.9 1024.52   437.9  1021.8     443 1021.38     448 1020.97     453 1021.42
   458.1 1021.87   518.5 1034.73   538.6 1039.17   548.7 1041.85   558.7  1045.3
   578.9 1053.57     599 1062.85   628.8 1075.68   638.7 1080.61   648.6 1086.94
   658.6 1094.37   757.9 1173.13   817.5 1218.67   847.2 1241.84   916.8 1294.08
#Mann= 3 , 0 , 0
       0     .06       0     443    .045       0     453     .06       0
Bank Sta=443,453
XS Rating Curve= 0 ,0
Exp/Cntr=0.3,0.1

Type RM Length L Ch R = 1 ,2971.4  ,296.7,283.3,269.9
XS GIS Cut Line= 4
     1704369.584      174212.879     1704434.284      173986.429
     1704511.923       173727.63     1704541.038        173410.6
#Sta/Elev= 30
     9.8 1199.16    29.4 1186.86    68.7 1162.99   117.8 1131.47   176.6 1098.19
   225.7 1072.05   285.5 1039.49   315.6  1023.7   335.6 1014.59   345.6 1011.74
   350.6  1011.4   355.6 1011.06   360.6 1011.53   365.6 1012.01   375.6 1013.82
   455.7 1030.97   465.7 1033.71   475.7 1037.77   485.7 1043.43   525.6 1070.62
   555.4 1089.55   575.3 1100.35   605.2  1114.2   615.1 1119.16     635 1130.46
   664.9 1149.24   704.7 1175.46   724.6 1189.19   784.3  1231.9   824.1 1261.66
#Mann= 3 , 0 , 0
       0     .06       0   350.6    .045       0   360.6     .06       0
Bank Sta=350.6,360.6
XS Rating Curve= 0 ,0
Exp/Cntr=0.3,0.1

Type RM Length L Ch R = 1 ,2688.1  ,425.9,439.5,453.1
XS GIS Cut Line= 4
     1704744.843      174361.688     1704799.838      174022.014
     1704702.788      173776.155     1704649.873      173421.909
#Sta/Elev= 30
     9.8 1164.87    29.5 1159.61      59 1150.55     177  1110.4   196.6    1103
   226.1 1090.65   265.4 1072.05   294.9 1059.21   363.7 1035.98   412.6 1016.78
   461.6 1004.18   471.4 1002.15   476.2 1002.13   481.2  1002.1   486.2 1003.42
   490.9 1004.65   510.5 1013.17   539.9 1024.32     579 1041.62   608.4 1056.67
   658.2 1086.35   668.1  1091.3     698 1102.85   727.8 1117.22   777.6 1139.94
   797.5 1150.28   827.3 1167.98   857.2  1186.8   936.7 1241.02   966.6 1262.32
#Mann= 3 , 0 , 0
       0     .06       0   476.2    .045       0   486.2     .06       0
Bank Sta=476.2,486.2
XS Rating Curve= 0 ,0
Exp/Cntr=0.3,0.1

Type RM Length L Ch R = 1 ,2248.6  ,458.2,461.4,464.5
XS GIS Cut Line= 4
     1704945.197      174433.276     1705087.752      174115.829
       1705164.2      173866.138     1705302.817      173589.389
#Sta/Elev= 30
     9.9  1241.9    39.8  1222.1    89.5 1188.04   198.8  1109.5   208.8 1102.62
   228.7 1090.88   268.4 1070.08   308.2 1050.04     338 1036.23   368.1 1023.26
   408.2 1008.03   458.5  992.25   463.5  991.74   468.5  991.23   473.5  991.97
   478.6  992.74   498.6   999.5   558.9 1016.36     589 1027.13   599.1 1031.38
   619.1 1041.26     659 1063.68     679 1073.37     689 1077.32   728.9    1091
   748.9 1098.79   768.9 1107.26   828.8 1135.47   898.7 1170.08   918.6 1178.31
#Mann= 3 , 0 , 0
       0     .06       0   463.5    .045       0   473.5     .06       0
Bank Sta=463.5,473.5
XS Rating Curve= 0 ,0
Exp/Cntr=0.3,0.1

Type RM Length L Ch R = 1 ,1787.2  ,541.6,532.4,523.2
XS GIS Cut Line= 4
     1705332.579      174603.309     1705485.656      174300.223
     1705599.068      174045.862     1705699.555      173760.069
#Sta/Elev= 30
      10 1272.73   119.8 1185.68   179.8 1139.53   199.7 1124.69   209.7 1118.06
   219.7 1112.18   239.7 1101.32   259.7 1089.23   289.6 1068.96   359.4 1019.44
   379.3 1006.57   389.3 1001.14   399.2  996.53   429.1   984.9     449  976.56
   453.9  976.06   458.9  975.54   463.9  976.54   468.9  977.54   488.7  985.32
   508.6   992.6   598.2 1024.78   678.6 1055.44   729.1 1075.27   739.2 1080.32
   749.3 1086.39   769.5 1099.49   799.8 1119.63   850.3 1152.54     921 1200.51
#Mann= 3 , 0 , 0
       0     .06       0   453.9    .045       0   463.9     .06       0
Bank Sta=453.9,463.9
XS Rating Curve= 0 ,0
Exp/Cntr=0.3,0.1

Type RM Length L Ch R = 1 ,1254.8  ,577.3,592.5,607.5
XS GIS Cut Line= 4
     1705970.686      174725.653     1706055.015      174406.978
      1706045.31      174115.829     1706052.682      173813.814
#Sta/Elev= 30
      10 1047.76    79.9 1033.11   149.8 1017.03   169.8 1013.83   219.8 1007.37
   269.7  999.02   319.7  989.22     400  972.11     410  970.37   430.1  969.18
   440.1  967.66   455.2  963.62   460.2  962.61   465.2  963.49   470.3  964.37
   480.3  967.99   490.4   969.8   510.5  971.34   520.5  973.68   530.5  977.01
   560.7  989.07     631 1020.82   671.3 1037.82   681.4 1042.56   701.5 1054.23
   721.7 1066.79   792.1 1115.12   822.4    1135   852.6  1152.3   923.1 1189.42
#Mann= 3 , 0 , 0
       0     .06       0   455.2    .045       0   465.2     .06       0
Bank Sta=455.2,465.2
XS Rating Curve= 0 ,0
Exp/Cntr=0.3,0.1

Type RM Length L Ch R = 1 ,662.3   ,374.7,376.2,377.8
XS GIS Cut Line= 4
      1706220.78      174881.674     1706452.919      174636.663
     1706637.314      174436.093     1706702.418       174099.99
#Sta/Elev= 30
     9.9 1131.84   148.9 1053.88   168.8 1042.13   248.2  989.64   258.1  982.61
     278  966.36   287.9  960.43   297.8  957.73   337.5  951.07   347.6  950.38
   377.9  950.25   408.2  951.42   418.2  950.65   443.5  945.44   448.5  944.84
   453.5  944.97   488.9  948.74     499  950.94   519.2  957.23   529.2  961.67
   549.4  973.31   559.5  980.51   599.9 1011.57     610 1018.56   630.1 1027.34
   700.6 1052.93   730.8 1063.03     761 1071.68     902 1107.58   952.3 1122.18
#Mann= 3 , 0 , 0
       0     .06       0   443.5    .045       0   453.5     .06       0
Bank Sta=443.5,453.5
XS Rating Curve= 0 ,0
Exp/Cntr=0.3,0.1

Type RM Length L Ch R = 1 ,286.1   ,182.4,173,163.3
XS GIS Cut Line= 4
      1706460.52      175132.724     1706669.664      174931.047
     1706902.583      174714.303     1707064.333      174316.398
#Sta/Elev= 30
      10 1142.25    60.1 1122.35    90.2 1104.72   130.2 1085.35   190.4 1054.64
   290.5  982.48   320.4  966.04   350.2  948.62   360.1  944.48   370.1   942.9
     390  943.86   399.9  943.51   409.9  941.77   429.7  937.03   434.7  936.47
   439.7   935.9   444.7  935.97   499.3  939.26   568.9  944.52   618.7  944.72
   628.7  945.16   648.7  947.41   668.6  951.56   708.6  963.39   728.6  968.38
   778.5  976.97   828.5  987.15   908.4  999.96   968.3 1014.78  1038.2 1027.25
#Mann= 3 , 0 , 0
       0     .06       0   434.7    .045       0   444.7     .06       0
Bank Sta=434.7,444.7
XS Rating Curve= 0 ,0
Exp/Cntr=0.3,0.1

Type RM Length L Ch R = 1 ,113.1   ,78.8,77,75.3
XS GIS Cut Line= 4
     1706572.614      175173.672     1706886.408      175018.392
     1706941.403      174863.112     1707057.863      174419.918
#Sta/Elev= 30
      10 1074.67      50 1063.55      60 1059.78      70 1053.74      90 1037.73
     110 1019.91     120    1010     140  984.92     150  975.03   160.1  967.86
   190.1  951.32   200.1  946.44   210.1   943.2   280.1  941.24   398.6   943.5
   427.6  940.17   451.7  933.16   456.7  932.08   461.7  932.26   466.4  932.44
   495.5  940.32   514.8  943.73   534.8  944.39   574.6  940.25   604.5   939.9
   684.2  946.14     744  952.88   773.8  957.16   863.5  973.45   973.1  996.17
#Mann= 3 , 0 , 0
       0     .06       0   451.7    .045       0   461.7     .06       0
Bank Sta=451.7,461.7
XS Rating Curve= 0 ,0
Exp/Cntr=0.3,0.1

Type RM Length L Ch R = 1 ,36.2    ,32.3,36.2,40.1
XS GIS Cut Line= 4
     1706625.288      175231.733     1706971.473      175024.755
     1707046.571        174755.5     1707075.877      174422.138
#Sta/Elev= 30
    10.1 1042.37    30.3  1028.8   100.8  976.12   131.1  954.66   141.2  948.54
   151.3  944.54   161.3  942.73   171.4  942.16   252.1  941.01   292.4  941.29
   373.1   944.3   383.2  943.83   403.3  941.22   463.2  937.51   473.2  936.37
   483.2  934.01   503.2  927.74   508.2  927.73   513.2  927.72   518.2  928.04
   543.1  929.01     613  927.77   662.9  928.11   702.6   929.8   732.1  932.58
   830.5  947.73   869.9   954.9   909.3  963.38   938.8  970.42  1017.5  991.25
#Mann= 3 , 0 , 0
    10.1     .06       0   508.2    .045       0   518.2     .06       0
#XS Ineff= 2 , 0
                          534.47          947.87
Permanent Ineff=
       F       F
Bank Sta=508.2,518.2
XS Rating Curve= 0 ,0
Exp/Cntr=0.3,0.1
Stream Node=Greenbrier Fork ,Main            , 0 , 0 ,Upstream end
Stream Node=Greenbrier Fork ,Main            , 0 , 1 ,Downstream end

Chan Stop Cuts=-1
Use User Specified Reach Order=0
